--- cnlyfrk.prj (project) ---

Proj Title=cnlyfrk
Current Plan=p01
Default Exp/Contr=0,0
English Units
Geom File=g01
Flow File=f01
Plan File=p01
BEGIN DESCRIPTION:
END DESCRIPTION:
DSS Export Rating Curves= 0
DSS Export Rating Curve Sorted= 0
DSS Export Volume Flow Curves= 0
DXF OffsetX= 0
DXF OffsetY= 0
DXF ScaleX= 0
DXF ScaleY= 0

--- cnlyfrk.p01 (plan) ---

Plan Title=Floodplain
Program Version=4.00
Geom File=g01
Flow File=f01
K Sum by GR=0
Std Step Tol=0.01
Critical Tol=0.01
Num of Std Step Trials=20
Max Error Tol=0.3
Flow Tol Ratio=0.001
Split Flow NTrial=30
Split Flow Tol=0.02
Split Flow Ratio=0.02
Log Output Level=0
Friction Slope Method=1
Unsteady Friction Slope Method=2
Unsteady Bridges Friction Slope Method=1
Global Log Level=0
CheckData=False
Run HTab=0
Run UNet=0
Run PostProcess=0
UNET Theta=0
UNET Theta Warmup=0
UNET ZTol=0
UNET ZSATol=0
UNET MxIter=0
UNET MaxInSteps=0
UNET DtIC=0
UNET DtMin=0
UNET MaxCRTS=0
UNET WFStab=0
UNET SFStab=0
UNET WFX=0
UNET SFX=0
UNET DSS MLevel=0
UNET DZMax Abort=0
UNET Convert EG Bridges=0
UNET Use Existing IB Tables=0
UNET Froude Limit=0
UNET Froude Power=0
Write IC File=0
Echo Input=False
Echo Output=False
Write Detailed=0

--- cnlyfrk.f01 (steady flow) ---

Flow Title=NFF Regression Equation
Program Version=4.00
Number of Profiles= 1
Profile Names=P100yr
River Rch & RM=cnlyfrk,Main            ,13206.1
     352
River Rch & RM=cnlyfrk,Main            ,13010.4
     363
River Rch & RM=cnlyfrk,Main            ,11260
     397
River Rch & RM=cnlyfrk,Main            ,10925.5
     543
River Rch & RM=cnlyfrk,Main            ,9765
     577
River Rch & RM=cnlyfrk,Main            ,6828.5
     631
River Rch & RM=cnlyfrk,Main            ,6489.7
     824
River Rch & RM=cnlyfrk,Main            ,4331.6
     880
River Rch & RM=cnlyfrk,Main            ,111.1
     973
Boundary for River Rch & Prof#=cnlyfrk,Main            , 1
Up Type= 0
Dn Type= 3
Dn Slope=0.022
DSS Import GetInterval= 0
DSS Import GetPeak= 0
DSS Import FillOption= 0

--- cnlyfrk.g01 (geometry) ---

Geom Title=USGS 10m DEM
Program Version=4.00

River Reach=cnlyfrk         ,Main
Reach XY= 30
      1656059.28      212022.881     1655721.081      211434.161
     1655115.902      210790.199     1654813.581      210356.822
     1654670.963      210227.057     1654315.638      210096.314
     1654161.807      210090.651      1653753.07      209860.677
     1652982.024      209710.295     1652882.914      209625.278
     1652485.429      209607.242     1652141.528       209728.56
     1651339.757      210326.193      1650842.53      210485.508
     1650318.292      210498.164     1649669.724      210354.363
     1649442.229      210375.666     1649284.727      210284.193
     1649199.067      210296.996     1648991.972      210477.006
     1648734.265       210551.22      1648622.39      210634.211
     1648514.303      210815.261     1648015.509      211368.619
     1647883.531      211464.592     1647005.958      211935.043
     1646552.074      212130.576      1646120.93      212527.911
      1645686.72      213181.904     1645394.958      213361.115

Type RM Length L Ch R = 1 ,13206.1 ,195.4,195.7,196
XS GIS Cut Line= 4
     1656355.332      211836.119     1656140.329      211921.222
     1655984.574      212021.065     1655714.998      212240.719
#Sta/Elev= 30
    10.1 1245.01    40.2  1224.6    60.3 1205.96    80.4 1192.99   130.7 1164.25
   150.8 1148.13   201.1 1122.68   211.1 1116.13   221.2 1106.26   270.2 1078.16
   289.7 1071.88   318.9 1072.85   347.8 1067.69   357.8  1067.6   367.8 1069.32
   377.3 1072.73     387  1081.6     456  1119.1   485.8 1123.25   495.7 1128.26
   515.6 1143.55   545.4 1161.67   565.3 1165.07   575.2 1170.45     605 1188.65
   664.6 1229.43   714.3 1244.74   734.2 1253.12     754 1272.24     764 1276.73
#Mann= 3 , 0 , 0
       0     .06       0   347.8    .045       0   367.8     .08       0
Bank Sta=347.8,367.8
XS Rating Curve= 0 ,0
Exp/Cntr=0.3,0.1

Type RM Length L Ch R = 1 ,13010.4 ,156.2,160.9,165.5
XS GIS Cut Line= 4
     1656261.023      211689.171     1656064.652      211739.906
     1655860.972      211867.205     1655636.326      212114.316
#Sta/Elev= 30
     9.7  1228.5    38.6 1211.32    48.3 1201.73    57.9 1194.44   125.6 1159.67
   135.2  1150.4   193.2 1120.76   212.8 1106.04   272.9 1074.84   292.9 1066.76
   332.9 1066.21   352.9 1064.66   362.9 1062.91   372.9 1063.47     403 1077.82
     413 1080.98     443 1085.38   453.1 1088.49   554.3 1159.12   574.6 1161.61
   584.7 1164.58   655.5 1218.07   665.6 1227.67   675.8 1238.96   685.9 1246.74
     696 1253.24   706.1 1257.03   726.4 1273.34   756.7 1300.91     777 1326.54
#Mann= 3 , 0 , 0
       0     .06       0   352.9    .045       0   372.9     .08       0
Bank Sta=352.9,372.9
XS Rating Curve= 0 ,0
Exp/Cntr=0.3,0.1

Type RM Length L Ch R = 1 ,12849.5 ,176.4,174.3,172.1
XS GIS Cut Line= 4
      1656242.38      211458.881     1655934.229      211652.983
       1655813.6      211700.138     1655626.077      212081.763
#Sta/Elev= 30
    10.1 1203.34    60.7 1179.11    70.8 1179.88      91 1173.65   141.6 1155.44
   161.9 1145.41   222.6 1134.71   242.8  1127.1   313.6 1108.72   374.2 1064.55
  440.04 1059.48   453.9 1058.71  458.04  1059.6   463.8 1060.87   483.7 1080.56
   493.7 1084.82   574.7 1086.89   594.9 1090.18   605.1 1096.85   615.2 1107.83
   655.7 1136.37   686.1 1149.32   706.3 1152.59   716.4 1157.91   736.7 1173.38
   767.1 1201.31   787.3 1210.23   827.8 1237.97   898.7 1291.48   918.9  1310.5
#Mann= 3 , 0 , 0
    10.1     .06       0  440.04    .045       0  458.04     .08       0
Bank Sta=440.04,458.04
XS Rating Curve= 0 ,0
Exp/Cntr=0.3,0.1

Type RM Length L Ch R = 1 ,12675.3 ,198.4,193.6,188.7
XS GIS Cut Line= 4
     1656204.228      211352.118     1655916.681      211459.948
     1655705.014      211563.785     1655433.664      211876.182
#Sta/Elev= 30
     9.9 1263.74    39.6 1252.17    79.3 1243.51    99.1 1235.18   118.9 1219.06
   168.4  1188.7   178.3 1180.88   188.2 1169.24   247.7 1135.57   267.5 1120.91
   336.6 1087.42     366 1066.33   385.7 1059.17  450.04  1054.9   464.3 1054.04
  470.03 1055.04   483.9 1061.87   513.4  1084.3   603.4 1087.89   633.7 1095.48
   653.9 1103.65   694.3 1128.83   714.4  1129.9   724.5 1133.31   754.8 1151.03
     775 1157.83     886 1217.07   896.1 1221.12   906.2 1219.68   956.7  1242.5
#Mann= 3 , 0 , 0
     9.9     .06       0  450.04    .045       0  470.03     .08       0
Bank Sta=450.04,470.03
XS Rating Curve= 0 ,0
Exp/Cntr=0.3,0.1

Type RM Length L Ch R = 1 ,12481.7 ,234.7,231.9,229.2
XS GIS Cut Line= 4
     1656034.699      211028.526     1655799.569      211269.646
     1655598.885      211422.406     1655311.338      211793.821
#Sta/Elev= 30
     9.9 1341.37    39.6 1320.55    49.5 1315.68     109 1261.33   158.5 1223.21
   188.2 1211.92   237.7 1176.83   257.5 1157.87   297.2 1132.34     317 1123.85
   336.8  1110.9     357 1093.12   407.4 1061.68   427.6 1052.19   498.3 1049.03
   508.3 1048.54   518.3 1050.18   538.6 1071.63   548.6  1076.1     619 1086.86
   668.9  1098.7   718.9  1117.8   758.9 1122.27   828.9 1148.56   848.8 1159.49
   888.8 1168.73   948.8 1175.83   968.8 1183.11  1028.7 1187.07  1058.7 1193.35
#Mann= 3 , 0 , 0
       0     .06       0   498.3    .045       0   518.3     .08       0
Bank Sta=498.3,518.3
XS Rating Curve= 0 ,0
Exp/Cntr=0.3,0.1

Type RM Length L Ch R = 1 ,12249.8 ,100,101.3,102.6
XS GIS Cut Line= 4
     1655899.819      210817.515     1655626.471      211090.863
     1655417.023      211289.661     1655012.327      211623.358
#Sta/Elev= 30
     9.9 1276.57    19.8 1268.17    49.6 1255.41   148.7 1200.07   168.5 1195.59
   198.2 1178.69   277.5 1148.59   426.4 1071.93   446.3 1066.42   496.1    1045
   545.9 1042.42   555.9 1041.99   565.9 1042.95   575.8 1044.89   605.6  1065.7
   665.4 1073.13   695.5 1084.05     756 1093.19   836.7  1152.2   856.9 1162.29
     867 1173.93   947.7 1240.18   957.8 1252.57   967.9 1261.25     978 1269.18
   998.1 1279.21  1038.5 1311.88  1048.6 1324.19  1068.7  1341.2  1199.9 1408.78
#Mann= 3 , 0 , 0
     9.9     .06       0   545.9    .045       0   565.9     .08       0
#XS Ineff= 2 , 0
       0     526                       0
Permanent Ineff=
       F       F
Bank Sta=545.9,565.9
XS Rating Curve= 0 ,0
Exp/Cntr=0.3,0.1

Type RM Length L Ch R = 1 ,12148.5 ,149.8,153.5,157.2
XS GIS Cut Line= 4
     1655780.999      210752.179     1655529.341      211051.994
     1655387.978      211173.163      1655010.49      211421.714
#Sta/Elev= 30
      10 1318.64    80.3 1250.68    90.3 1243.89   100.4 1240.86   160.6 1202.07
   180.7 1182.93   210.8 1162.55   230.8 1154.77     261 1136.92     281 1121.52
   361.3 1084.22   391.4 1064.67   430.6 1045.98   450.2 1041.48     499  1040.1
     509 1038.39     519 1039.46     558 1063.41   567.8 1065.95   607.8 1065.42
   688.1 1070.67   708.2 1076.99   768.5 1124.27   808.6 1146.01   828.7 1165.05
     899  1217.9   919.1 1236.11   939.2 1249.43   959.3 1255.52  1029.6  1297.1
#Mann= 3 , 0 , 0
       0     .06       0     499    .045       0     519     .08       0
Bank Sta=499,519
XS Rating Curve= 0 ,0
Exp/Cntr=0.3,0.1

Type RM Length L Ch R = 1 ,11995   ,154.5,150.9,147.4
XS GIS Cut Line= 4
     1655708.213      210675.082     1655483.567      210923.691
     1655272.399      211056.981     1654891.998      211331.049
#Sta/Elev= 30
     9.9 1305.84    49.3 1276.39      69 1266.42    78.8  1255.8    88.7 1247.74
   177.4  1182.3   266.1 1123.85   285.8 1105.07   295.7 1098.47   315.4  1089.4
     355 1063.54     365 1056.72     375  1046.4     385 1039.73     405 1035.41
   464.9 1037.52   504.9 1033.06   514.9  1032.3   524.9 1033.81   554.8 1047.93
   594.8 1052.47   714.5  1092.9   774.3 1124.66   794.3 1132.15   814.2 1147.26
   844.1 1162.95   933.9 1204.91   973.8 1221.32   993.8 1235.94  1053.6 1265.02
#Mann= 3 , 0 , 0
     9.9     .06       0   504.9    .045       0   524.9     .06       0
#XS Ineff= 2 , 0
       0     454                       0
Permanent Ineff=
       F       F
Bank Sta=504.9,524.9
XS Rating Curve= 0 ,0
Exp/Cntr=0.3,0.1

Type RM Length L Ch R = 1 ,11844   ,123.4,125.4,127.5
XS GIS Cut Line= 4
     1655596.139      210595.281     1655283.897      210862.474
     1655162.728      210965.001     1654853.593      211236.854
#Sta/Elev= 30
      10 1275.96    30.1 1268.88    50.1 1251.41   120.3 1202.27   140.3  1183.7
   170.4 1168.07   200.5 1146.27   210.5 1138.34   230.5 1116.89   300.7 1061.22
   310.7 1048.52   330.8 1033.48   350.8 1029.04   430.8 1033.44   460.6 1033.26
  476.97 1029.73   480.4 1028.63  492.07 1029.76   549.8 1061.01   559.8 1064.02
   589.8  1065.8     640 1083.15   670.1 1097.76   690.2 1114.11   760.5 1154.81
   780.5 1172.17   860.9 1215.18   880.9 1230.59   951.2 1265.32   981.3 1285.51
#Mann= 3 , 0 , 0
      10     .06       0  476.97    .045       0  492.07     .06       0
#XS Ineff= 2 , 0
       0     440                       0
Permanent Ineff=
       F       F
Bank Sta=476.97,492.07
XS Rating Curve= 0 ,0
Exp/Cntr=0.3,0.1

Type RM Length L Ch R = 1 ,11718.6 ,147,147,146.9
XS GIS Cut Line= 4
     1655559.946      210535.801     1655317.328      210693.054
     1655070.217      210869.775     1654791.656      211217.229
#Sta/Elev= 30
      10  1278.6    29.9 1269.94    69.8 1243.27    89.7 1225.15   109.7 1216.72
   159.5 1185.07   179.5 1167.32   259.2 1111.58   299.2  1085.9   329.6 1058.82
   349.9 1031.18     360 1028.15   461.3 1028.96   491.8 1023.88   501.8 1022.48
   511.8 1024.12   532.2 1040.11   562.5 1056.11   572.7 1060.08     603 1062.82
   643.5 1080.89   704.3 1117.91   714.4 1128.07   805.5 1187.84   825.7 1203.61
   835.8 1207.12   916.8 1251.34     937 1266.36    1018 1305.73  1038.3 1321.16
#Mann= 3 , 0 , 0
       0     .06       0   491.8    .045       0   511.8     .06       0
Bank Sta=491.8,511.8
XS Rating Curve= 0 ,0
Exp/Cntr=0.3,0.1

Type RM Length L Ch R = 1 ,11571.7 ,162.9,164.6,166.2
XS GIS Cut Line= 4
     1655446.231      210417.088     1655133.694      210644.089
     1655014.162      210729.626     1654662.146       211066.29
#Sta/Elev= 30
     9.9 1270.31    39.6 1249.69    59.4 1231.21    89.1 1210.86   108.9 1201.61
   128.8 1188.12   148.6  1169.7   217.9  1126.1   237.7 1108.14   267.4 1091.43
     307 1057.79   326.8 1033.97   336.8 1027.76   445.1 1025.13   474.3 1018.29
   484.3 1016.54   494.3 1019.34   533.3 1045.25     573  1054.2   592.9 1070.53
   662.5 1112.18   682.4  1128.8   702.3 1138.98   761.9 1178.45   801.7 1210.26
   861.3 1242.74   881.2 1260.42   920.9 1287.09   990.5 1327.46  1020.4 1341.13
#Mann= 3 , 0 , 0
       0     .06       0   474.3    .045       0   494.3     .06       0
Bank Sta=474.3,494.3
XS Rating Curve= 0 ,0
Exp/Cntr=0.3,0.1

Type RM Length L Ch R = 1 ,11407.1 ,147,147.1,147.2
XS GIS Cut Line= 4
     1655399.273       210309.87     1655150.776      210448.319
     1654870.328      210622.267     1654586.331      211041.163
#Sta/Elev= 30
     9.8 1289.71    19.6 1274.97    29.4 1266.16    88.3 1223.41   107.9 1204.55
   166.8 1167.91   186.4 1150.03     255 1110.27   284.5 1085.32   334.5 1049.94
   354.5 1027.56   374.5 1021.07   474.5 1023.59   507.6 1012.07   514.5 1009.46
  520.67 1011.83   544.5 1031.19   584.5  1047.5   604.5 1065.01   634.7 1079.54
   675.2 1104.29   725.8 1140.52   756.2 1155.21   816.9 1193.44   837.2  1210.8
   897.9 1244.58   928.3 1264.55   958.6 1290.05  1039.6  1331.5  1120.6 1360.93
#Mann= 3 , 0 , 0
     9.8     .08       0   507.6    .045       0  520.67     .08       0
Bank Sta=507.6,520.67
XS Rating Curve= 0 ,0
Exp/Cntr=0.3,0.1

Type RM Length L Ch R = 1 ,11260   ,90.5,90.6,90.7
XS GIS Cut Line= 4
     1655379.337      210288.783     1654977.973      210383.093
     1654832.122      210473.016     1654640.213      210670.408
#Sta/Elev= 30
    10.1 1275.78    60.3 1237.65    70.4 1224.73    80.4 1216.64   140.8 1176.29
   160.9 1159.33   211.2 1134.34   231.3 1120.17   261.5 1107.94   281.6 1096.39
   291.6 1088.07   301.7 1074.03     362 1024.79   372.1 1020.01   382.1 1019.47
   482.8  1022.2     503 1018.28  529.95 1005.68   533.2 1004.28  544.87 1005.76
   573.6 1027.89   603.3 1041.59   642.6 1069.57   652.5 1073.08   721.3 1115.08
   770.5 1150.88   790.1 1158.57   819.6 1177.33   839.3 1194.29   858.9 1207.08
#Mann= 3 , 0 , 0
    10.1     .08       0  529.95    .045       0  544.87     .08       0
Bank Sta=529.95,544.87
XS Rating Curve= 0 ,0
Exp/Cntr=0.3,0.1

Type RM Length L Ch R = 1 ,11169.4 ,113.7,109.1,104.5
XS GIS Cut Line= 4
     1655383.225      210248.254     1655047.753      210234.775
     1654739.238      210423.478     1654570.005      210627.157
#Sta/Elev= 30
     9.9  1269.3    69.1 1238.31    88.9 1221.21   138.2 1189.94     158 1174.47
   227.1    1141     237 1132.53   266.6 1119.08   296.2 1098.03   345.8 1079.67
     386 1047.15     396 1031.16   406.1 1022.47   416.1 1018.27   426.2 1017.46
   546.7 1020.96  589.85  999.58   596.9  998.33   601.8   999.5     607 1000.74
   647.2 1026.26   697.4 1047.51   746.4 1080.87   795.5 1110.66   815.1 1117.34
   834.7 1129.22   854.3  1145.2   913.2 1186.39   932.8 1191.76   962.2 1205.25
#Mann= 3 , 0 , 0
     9.9     .08       0  589.85    .045       0   601.8     .08       0
Bank Sta=589.85,601.8
XS Rating Curve= 0 ,0
Exp/Cntr=0.3,0.1

Type RM Length L Ch R = 1 ,11060.4 ,153.1,134.9,116.7
XS GIS Cut Line= 4
      1655370.89      210230.222     1654855.146      210197.599
     1654701.355      210335.856     1654538.243      210604.602
#Sta/Elev= 30
    10.1 1251.25    60.8 1224.38    70.9  1214.2   101.3 1196.82   141.9 1178.71
     152 1170.45   212.8 1140.47   222.9 1131.47   253.3 1116.78   283.7 1094.54
   354.6 1068.86   364.8 1062.48   374.9 1049.15     385 1041.09   425.6 1019.18
     456 1015.37   516.8 1019.19   575.9 1016.39   644.6  995.63   654.6   994.2
   664.6  996.31     694 1009.96   713.7 1015.34   792.3 1062.82     812    1069
   900.4 1124.13   929.9 1135.78     979 1170.46  1018.3 1185.26  1037.9 1185.67
#Mann= 3 , 0 , 0
       0     .08       0   644.6    .045       0   664.6     .08       0
Bank Sta=644.6,664.6
XS Rating Curve= 0 ,0
Exp/Cntr=0.3,0.1

Type RM Length L Ch R = 1 ,10925.5 ,130.5,134.4,138.3
XS GIS Cut Line= 4
      1654516.09      209514.409     1654665.854      210061.049
     1654626.915      210293.183      1654465.17      210601.698
#Sta/Elev= 30
    10.1 1342.71    40.5 1317.89    60.7 1310.42   151.8  1240.9   161.9 1240.42
   202.4 1211.65   263.1 1172.83   283.4 1166.62   364.4 1107.74   374.5 1102.55
   384.6 1100.84   485.8 1033.85   495.9 1033.23   536.4 1010.86     606 1005.98
   684.5  993.61  720.01  990.91   733.5     990  737.77  991.49   772.7 1004.51
   792.4 1014.14   812.1  1020.3   911.6 1078.18   921.6 1078.84   961.4 1103.35
  1011.2 1129.23  1031.1 1133.55  1070.9    1149  1120.6 1164.46  1150.5 1170.28
#Mann= 3 , 0 , 0
    10.1     .06       0  720.01    .045       0  737.77     .06       0
Bank Sta=720.01,737.77
XS Rating Curve= 0 ,0
Exp/Cntr=0.3,0.1

Type RM Length L Ch R = 1 ,10791.1 ,137.9,137.8,137.8
XS GIS Cut Line= 4
     1654503.135      209525.533     1654542.614      210092.488
     1654489.976      210250.402     1654375.927      210556.359
#Sta/Elev= 30
      10  1333.1    29.9  1315.5    49.9 1307.07   119.6 1250.71   129.6 1243.88
   149.6 1237.53   229.3 1182.02   239.3 1176.99   249.3 1174.91     339 1107.79
     349 1106.93   378.9 1081.95   448.7 1031.55   458.6 1030.97   488.6 1011.72
   498.5 1008.07   528.4 1006.99   568.3 1000.44   617.3  988.21     666  984.05
     676  983.46     686  985.23   764.5 1032.86   774.4 1033.56   853.5 1077.46
   863.4 1081.36   873.3 1081.88   962.4 1119.62   982.1 1123.79  1061.3 1156.55
#Mann= 3 , 0 , 0
       0     .06       0     666    .045       0     686     .06       0
Bank Sta=666,686
XS Rating Curve= 0 ,0
Exp/Cntr=0.3,0.1

Type RM Length L Ch R = 1 ,10653.3 ,131.6,127,122.4
XS GIS Cut Line= 4
     1654481.644      209503.926     1654441.207      209972.688
     1654354.344      210224.292     1654218.059      210531.308
#Sta/Elev= 30
      10 1351.88      40 1326.19    60.1 1317.32   100.1 1280.45   130.1  1257.3
   140.1 1251.17   160.2 1245.85   180.2 1235.98   240.3 1192.56   270.3  1178.1
   340.4 1125.83   360.4  1107.6   370.4 1107.38   420.4 1053.17   450.5 1029.31
   500.1 1009.47   539.5 1004.15   569.1  993.57   578.9  993.33   598.7  985.78
   628.1  979.96   638.1  979.29   648.1  980.85   677.5  989.89   726.8 1019.44
   766.3 1039.11   786.1 1043.39     875 1083.81   894.8 1088.15  1072.6 1157.15
#Mann= 3 , 0 , 0
       0     .08       0   628.1    .045       0   648.1     .08       0
Bank Sta=628.1,648.1
XS Rating Curve= 0 ,0
Exp/Cntr=0.3,0.1

Type RM Length L Ch R = 1 ,10526.3 ,230.7,236.2,241.6
XS GIS Cut Line= 4
     1654421.735      209537.385     1654280.371      210003.419
     1654263.284      210130.801     1654129.687      210497.414
#Sta/Elev= 30
     9.9 1324.74    19.9 1323.45    29.8 1316.97    99.4 1260.34   119.3 1249.71
   129.2 1248.87   208.7  1189.6   228.6 1182.11     318 1112.08     328 1111.18
   417.4 1039.88   427.4 1034.26   437.3 1032.32   467.1 1008.32   477.1 1004.22
   506.8 1001.33   526.5  991.72   536.4  990.38     566  977.47     576  975.87
     586  976.65   635.5  995.04   645.5  996.55   735.6  1045.8   755.6 1051.17
   845.6 1099.72   865.7 1106.21   945.7 1148.73   965.7 1154.48  1005.7 1173.71
#Mann= 3 , 0 , 0
       0     .08       0     566    .045       0     586     .08       0
Bank Sta=566,586
XS Rating Curve= 0 ,0
Exp/Cntr=0.3,0.1

Type RM Length L Ch R = 1 ,10290.2 ,249.8,252.4,255
XS GIS Cut Line= 4
     1654418.373      209470.969     1654105.976      209875.665
     1654003.027      210156.112     1653985.277      210518.209
#Sta/Elev= 30
      10 1353.41    40.1 1348.72   110.3 1320.13   140.3 1299.04   170.4 1272.14
   200.5  1249.2   220.5 1241.65   290.7 1189.47   330.8 1165.13   340.8 1163.94
   441.1 1091.68   461.1 1083.66     561 1006.95   610.8 1000.93   630.7  990.36
   650.7   975.5  665.44   971.4   680.5  970.48  685.13  971.46   730.3  995.03
   790.1 1017.18   870.4 1062.76   900.6  1074.3   981.2 1120.97   991.3 1122.04
  1001.3 1126.79  1081.9 1168.98    1102 1174.19  1122.2 1187.12  1172.5 1226.92
#Mann= 3 , 0 , 0
      10     .08       0  665.44    .045       0  685.13     .08       0
Bank Sta=665.44,685.13
XS Rating Curve= 0 ,0
Exp/Cntr=0.3,0.1

Type RM Length L Ch R = 1 ,10037.8 ,277.7,272.8,267.8
XS GIS Cut Line= 4
      1654337.87       209526.39     1653936.502      209688.136
     1653770.264      210031.096     1653633.978      210248.254
#Sta/Elev= 30
    10.1 1319.86    30.2 1302.67    90.6  1262.4   100.6 1252.59   171.1 1215.85
   191.2 1200.73   251.6  1169.2   271.7 1154.59     322 1131.26   332.1 1124.36
   342.2 1113.22   402.5 1068.18   422.7 1045.81   432.7    1039   543.1 1000.65
   593.2   996.3   643.4  970.58   653.4   967.1   673.5  965.27   683.5  964.49
   693.5  966.87   743.7  980.28   773.7  993.08   783.8  993.59   803.8 1002.36
     873 1042.21   892.7 1048.57   991.4 1107.09  1011.1 1113.01  1070.2 1143.73
#Mann= 3 , 0 , 0
       0     .08       0   673.5    .045       0   693.5     .08       0
Bank Sta=673.5,693.5
XS Rating Curve= 0 ,0
Exp/Cntr=0.3,0.1

Type RM Length L Ch R = 1 ,9765    ,289.7,287.5,285.3
XS GIS Cut Line= 4
     1653541.125      209252.322     1653627.988      209614.751
     1653538.129      209962.204     1653479.721      210201.827
#Sta/Elev= 30
    10.1 1296.77    40.3  1274.4    90.7 1225.32   110.8 1216.83   161.2 1186.23
   211.5 1165.27   221.6 1164.89     272 1126.44   312.3 1083.73   322.3  1081.3
   372.7 1048.09   422.5 1011.69   462.4  995.73   492.3  993.42   522.2  979.61
   542.2  974.01   562.1  963.13     582  958.61     592  958.07     602  959.59
   621.9  967.47   651.8  971.81   671.8  979.41   731.6 1016.76   751.3 1022.92
   830.2 1075.33     850 1081.85   938.8 1140.93   958.5 1147.83   978.2 1160.96
#Mann= 3 , 0 , 0
       0     .08       0     582    .045       0     602     .08       0
Bank Sta=582,602
XS Rating Curve= 0 ,0
Exp/Cntr=0.3,0.1

Type RM Length L Ch R = 1 ,9477.5  ,246.6,247.7,248.8
XS GIS Cut Line= 4
     1653452.764      209217.876     1653326.962      209565.329
     1653279.037      209851.379     1653114.296      210108.973
#Sta/Elev= 30
      10 1289.34      30 1279.77    99.9 1227.45   119.8 1213.94   139.8  1206.1
   209.7 1157.64   269.7 1135.54   299.6 1119.28   329.6 1098.05   339.6 1096.02
   349.6 1088.73   389.5 1047.23   429.5 1000.03   439.5  994.73   479.5  985.79
   529.5  958.21   559.6   951.4   569.6  950.64   579.6  951.83   599.6  958.51
   649.6   966.2   679.3  975.01   708.9  989.31   758.2 1018.92   768.1  1018.7
   777.9  1022.4   856.8 1058.64   896.3 1067.51   935.7 1091.43   965.3 1104.54
#Mann= 3 , 0 , 0
       0     .06       0   559.6    .045       0   579.6     .08       0
Bank Sta=559.6,579.6
XS Rating Curve= 0 ,0
Exp/Cntr=0.3,0.1

Type RM Length L Ch R = 1 ,9229.8  ,110.8,117.4,124.1
XS GIS Cut Line= 4
     1653312.202      209169.131     1653066.558      209647.259
      1653036.95       209786.53     1652919.611      210027.787
#Sta/Elev= 30
      10 1267.85    49.8 1231.72    59.7 1229.99    69.7 1223.43   159.3 1154.91
   179.2  1145.1   278.7 1078.31   288.7 1077.21   298.6 1071.01   378.3 1015.03
   398.2 1007.79     428  988.55   457.9  985.25   487.8   974.4   507.7  970.35
     566  948.82     613  945.86     623  945.09     633  946.79   699.8  994.86
   709.7 1001.03   719.7 1002.13   759.4 1028.89   809.1 1066.71     819 1068.25
     829  1073.5   898.5 1117.03   918.4 1127.89   938.3 1135.29   948.2  1142.5
#Mann= 3 , 0 , 0
       0     .06       0     613    .045       0     633     .08       0
Bank Sta=613,633
XS Rating Curve= 0 ,0
Exp/Cntr=0.3,0.1

Type RM Length L Ch R = 1 ,9112.4  ,100.7,98.6,96.4
XS GIS Cut Line= 4
     1653249.143       209171.29     1652978.844      209614.022
     1652911.657      209744.317     1652844.082      210026.267
#Sta/Elev= 30
      10 1244.59    49.9 1211.28    59.9 1209.54    69.8 1203.46   149.6 1145.21
   159.6  1139.7   169.6 1138.13   199.5 1114.72   269.3  1068.5   289.3 1061.44
   309.2 1045.67   379.1  996.77     409  984.67   438.9   981.1   498.8  950.42
   538.3  943.15   567.6  943.99   596.7  940.72   606.7  940.46   616.7  942.41
   626.2  945.43   715.3 1021.56   725.3 1023.42   765.3 1051.61   815.3 1082.57
   835.3 1088.59   915.3 1137.03   925.3 1141.74   935.3 1143.54   955.3 1157.42
#Mann= 3 , 0 , 0
      10     .06       0   596.7    .045       0   616.7     .08       0
#XS Ineff= 2 , 0
       0     567                       0
Permanent Ineff=
       F       F
Bank Sta=596.7,616.7
XS Rating Curve= 0 ,0
Exp/Cntr=0.3,0.1

Type RM Length L Ch R = 1 ,9013.8  ,319.3,307.7,296
XS GIS Cut Line= 4
     1653186.535      209151.471     1652959.337      209424.819
     1652842.188      209705.266     1652746.339      210095.763
#Sta/Elev= 30
     9.9 1240.38    69.1 1199.79      79 1198.13   108.6 1180.16   187.6 1124.03
   197.5 1122.67   207.3 1117.18   276.5 1069.42   306.1 1046.39   325.8 1039.37
     396  985.94   406.1  982.17   436.5  979.69   517.5  942.63   558.2   935.7
   568.2  934.63   578.2  935.07   608.7  945.33   639.1   965.2   659.4  973.01
   739.8 1033.52   759.9 1041.24   840.3 1091.01   850.4  1092.6   860.4 1097.51
   940.8 1148.52   960.9 1155.93  1021.3 1199.61  1051.4 1224.48  1061.5 1225.12
#Mann= 3 , 0 , 0
       0     .08       0   558.2    .045       0   578.2     .08       0
Bank Sta=558.2,578.2
XS Rating Curve= 0 ,0
Exp/Cntr=0.3,0.1

Type RM Length L Ch R = 1 ,8706.2  ,159.2,150.9,142.7
XS GIS Cut Line= 4
     1652416.395       209151.98     1652555.676      209403.584
     1652575.145      209712.098     1652656.018      210068.537
#Sta/Elev= 30
     9.9 1162.86    89.2 1113.43   109.1 1106.64   218.2 1030.27     238 1022.99
   257.8 1008.74   307.5  981.86   317.5  977.65   327.5  975.84   347.4  975.13
   367.4  970.54   427.2  946.94   447.1   943.1     487  927.67     497  926.88
     507  927.91   526.9  933.07   546.9  945.04   556.8  946.79   596.7  977.34
   646.1 1013.45     656 1014.27   744.9 1077.93   754.8 1082.55   764.6 1084.96
   863.4 1152.04   873.3 1153.47   883.2 1158.38   912.8 1179.68   962.2 1220.73
#Mann= 3 , 0 , 0
       0      .1       0     487    .045       0     507      .1       0
Bank Sta=487,507
XS Rating Curve= 0 ,0
Exp/Cntr=0.3,0.1

Type RM Length L Ch R = 1 ,8555.2  ,154.5,153.6,152.7
XS GIS Cut Line= 4
      1652304.39      209200.288     1652389.829      209548.259
     1652456.627      209711.371     1652571.582      210039.148
#Sta/Elev= 30
      10 1132.65    29.9 1127.07   119.4 1070.79   139.3 1064.27   159.2 1050.64
   179.2  1033.6   189.1 1026.87   228.9 1003.41   248.8  997.35   288.6  973.65
   298.6  971.51   318.5  970.69   348.4  960.32   358.3  958.93   441.8  922.99
   446.4  921.71   461.6  922.52   485.6  927.05   495.4  931.66   574.3  986.62
   584.2  988.88   594.1  993.69   683.4 1053.35   693.4 1054.52   703.3 1060.32
   733.1 1080.45   762.8 1103.66   802.5    1131   812.4 1131.75   881.9 1174.94
#Mann= 3 , 0 , 0
      10      .1       0   441.8    .045       0   461.6      .1       0
Bank Sta=441.8,461.6
XS Rating Curve= 0 ,0
Exp/Cntr=0.3,0.1

Type RM Length L Ch R = 1 ,8401.7  ,235.9,231.9,227.8
XS GIS Cut Line= 4
     1652040.487      209198.407     1652194.744       209494.94
     1652322.044      209774.999     1652525.723      210068.537
#Sta/Elev= 30
    10.1 1133.49    70.9 1116.72    91.2  1107.6   121.5 1098.34   162.1 1081.37
   192.5 1064.68     233 1034.39   243.1    1032   283.6 1008.85   324.1  989.36
     364  974.31   383.9  969.82   413.6  966.23   463.3   945.7   483.1  941.61
   532.7  919.09   542.7  918.39   552.7  919.39   582.3  925.44   592.3  931.23
   602.2  932.77   612.1  937.86   721.3 1006.83   741.1 1015.16   860.2 1092.72
   870.2 1094.64     890 1109.07   939.6 1140.24   989.2 1170.62   999.2 1174.97
#Mann= 3 , 0 , 0
       0      .1       0   532.7    .045       0   552.7      .1       0
Bank Sta=532.7,552.7
XS Rating Curve= 0 ,0
Exp/Cntr=0.3,0.1

Type RM Length L Ch R = 1 ,8169.8  ,233.5,230.9,228.4
XS GIS Cut Line= 4
     1651780.361      209367.995     1651995.902      209662.761
     1652115.905      209843.349     1652367.563      210131.125
#Sta/Elev= 30
     9.9 1180.42   128.3 1124.07   138.2 1120.81     148 1121.42   207.3 1093.14
   236.9 1072.05   276.3 1037.08   286.2 1033.39   325.7  987.65   345.4  968.87
   355.3  965.08   424.3  961.59   434.2  958.16   473.6   930.1   483.4  919.91
   493.1  913.37   503.1   912.5   513.1  913.14   562.3  917.03     582  922.68
   612.2  941.05   632.3  956.14   682.6  984.93   702.7  991.77   773.1 1043.17
   833.5 1081.26   853.6 1087.96     924 1134.01   944.2  1143.2   964.3 1147.46
#Mann= 3 , 0 , 0
       0      .1       0   493.1    .045       0   513.1      .1       0
Bank Sta=493.1,513.1
XS Rating Curve= 0 ,0
Exp/Cntr=0.3,0.1

Type RM Length L Ch R = 1 ,7938.9  ,181,181.2,181.5
XS GIS Cut Line= 4
     1651585.499      209520.668     1651777.198      209779.816
     1651968.896      210014.113     1652252.893      210308.761
#Sta/Elev= 30
    10.1 1099.44    30.2 1089.17    50.4 1084.03   171.2 1022.46   201.5 1014.33
   211.5 1010.13   261.9  987.71   282.1  975.87   312.3  966.55   332.4  962.37
   352.6  959.83   413.2  956.83   463.6  928.21   483.8  920.83   493.9  913.23
   504.1  909.31   514.1  908.95   524.1  909.62   564.5  914.41   625.1  926.38
     645  935.08   694.9  961.43   794.8  989.34   804.7  995.36   824.7 1002.34
   924.5 1024.51   944.5 1034.58   954.5 1037.19  1004.4 1045.19  1034.3 1051.77
#Mann= 3 , 0 , 0
       0      .1       0   504.1    .045       0   524.1      .1       0
Bank Sta=504.1,524.1
XS Rating Curve= 0 ,0
Exp/Cntr=0.3,0.1

Type RM Length L Ch R = 1 ,7757.7  ,167.2,165.6,164.1
XS GIS Cut Line= 4
     1651417.373      209689.623     1651651.943      209903.998
     1651805.734      210095.072     1652010.789      210461.685
#Sta/Elev= 30
     9.9 1145.82    29.8 1130.11    39.7 1119.43    49.7 1112.41    69.5 1100.12
    89.4 1091.45   129.1 1068.37     149 1052.92   168.8 1041.14   278.1  982.71
   347.2   953.8   376.6  938.83   406.1  919.76  440.04  907.17   445.3  906.37
   464.9  906.84   533.6  908.66   563.1  911.68   583.1   917.3   673.1  972.02
   703.1  985.42   723.1 1001.24   773.1 1035.14   803.1 1054.16   823.1 1061.37
   883.1 1098.99   913.1 1121.45   933.1 1133.98   953.1 1140.93   983.1 1159.43
#Mann= 3 , 0 , 0
     9.9      .1       0  440.04    .045       0   464.9      .1       0
Bank Sta=440.04,464.9
XS Rating Curve= 0 ,0
Exp/Cntr=0.3,0.1

Type RM Length L Ch R = 1 ,7592    ,254.3,254.7,255.2
XS GIS Cut Line= 4
     1651245.239       209888.82     1651529.791      210026.603
     1651721.489      210236.273      1651886.23      210573.243
#Sta/Elev= 30
     9.9 1161.51    59.3  1130.6      79 1113.85   128.4 1088.42   158.1 1070.52
     168 1060.78     247 1015.03   266.8  999.77   316.2  972.01   345.5  951.55
   365.1  934.11   384.7  926.17   404.3   910.1   414.1  903.68  420.64  902.42
   423.9  901.71  440.07  902.29   531.7  902.99   561.1  905.78   570.9  909.52
   600.2  926.55   649.6  970.48   659.5     976   669.3  977.64   777.9 1046.14
   797.7 1053.32   837.1 1082.56   906.2    1126   916.1 1127.56   975.3 1161.78
#Mann= 3 , 0 , 0
     9.9      .1       0  420.64    .045       0  440.07      .1       0
Bank Sta=420.64,440.07
XS Rating Curve= 0 ,0
Exp/Cntr=0.3,0.1

Type RM Length L Ch R = 1 ,7337.3  ,249.1,259.2,269.3
XS GIS Cut Line= 4
     1651173.703      209900.514     1651326.352      210177.412
      1651539.35       210418.81     1651844.647      210621.158
#Sta/Elev= 30
     9.9 1192.42    29.6 1180.97    39.5 1178.23   138.3 1111.93   158.1 1103.26
   197.6 1075.39   237.1 1045.38   266.8 1017.55   276.7 1013.93   286.5 1007.18
   346.4   949.7   406.7  913.42   426.9  906.14   436.9  897.99     447  893.61
     457  892.79     467  893.45   587.8  903.58   607.9     918   697.5  970.94
   717.3  987.91     747 1006.39   766.8 1014.37   786.6  1026.6   816.3 1050.79
   885.6 1095.49   905.4 1111.54   964.8 1146.31   984.6 1155.25  1004.4 1168.14
#Mann= 3 , 0 , 0
       0      .1       0     447    .045       0     467      .1       0
Bank Sta=447,467
XS Rating Curve= 0 ,0
Exp/Cntr=0.3,0.1

Type RM Length L Ch R = 1 ,7078.1  ,249,249.6,250.3
XS GIS Cut Line= 4
     1651152.385       209920.27     1651143.399      210269.221
      1651231.76      210532.806     1651052.043      211021.037
#Sta/Elev= 30
      10 1188.33    89.8 1126.72   109.7 1118.95   189.5 1053.77   219.4 1037.85
   299.2  979.85   309.2   974.4   319.1  973.32   388.8  934.42   408.6  918.22
   428.5  908.05   448.4  887.63  453.93  885.86   458.3  884.22  472.74   885.6
   517.9  888.99   707.1  891.87   717.1  895.45   737.1  911.05   757.1  918.25
   797.2  945.49   847.2  984.41   867.2   992.4   887.2 1008.36   947.2 1048.19
   967.2 1054.87  1057.3 1116.58  1067.3 1116.98  1077.3 1122.83  1147.3 1169.85
#Mann= 3 , 0 , 0
      10      .1       0  453.93    .045       0  472.74     .08       0
Bank Sta=453.93,472.74
XS Rating Curve= 0 ,0
Exp/Cntr=0.3,0.1

Type RM Length L Ch R = 1 ,6828.5  ,329.2,338.8,348.4
XS GIS Cut Line= 4
     1650848.364      209989.162     1650903.906       210326.51
     1650978.658      210570.247     1651017.597      211007.559
#Sta/Elev= 30
    10.1 1146.68    90.5 1085.14   100.6 1078.94   120.7 1070.25   160.9 1040.07
   211.2 1005.14   221.2 1004.71   271.5  971.02   311.7  948.43   321.8  947.46
   351.7  932.41   381.1  923.77   430.1  892.78   439.9  892.23   449.8  883.49
   459.4  878.04   469.4  877.39   479.4   878.3   596.8  885.52   646.7  913.17
   666.7  918.83   746.5  965.89   766.5  971.93   776.4  978.23   846.3 1029.67
   856.3  1034.7   866.2 1036.95     966 1109.49     976 1110.45  1035.9 1156.31
#Mann= 3 , 0 , 0
       0      .1       0   459.4    .045       0   479.4      .1       0
Bank Sta=459.4,479.4
XS Rating Curve= 0 ,0
Exp/Cntr=0.3,0.1

Type RM Length L Ch R = 1 ,6489.7  ,183.3,181.5,179.7
XS GIS Cut Line= 4
     1650641.689      210032.594     1650619.224      210380.046
     1650599.755      210609.186     1650716.571      210998.573
#Sta/Elev= 30
     9.9 1149.74    29.8 1139.42    39.8 1137.67    59.7 1128.54   129.3 1083.75
   149.2 1076.79     199 1042.81   238.8 1008.44   248.7 1004.92   288.5  952.29
   298.4  941.25   318.3  925.26   328.3  921.22   358.2  918.73   368.2  913.73
   418.2  877.47   428.2  871.95   438.2  870.89   448.2  871.14   558.1  877.68
   578.1  885.53   647.6  921.36   657.5  925.56   667.4  925.97   766.5  978.82
   786.4  985.77   875.6 1046.91   885.5 1048.85   895.4  1053.8   984.7 1118.67
#Mann= 3 , 0 , 0
       0      .1       0   428.2    .045       0   448.2      .1       0
Bank Sta=428.2,448.2
XS Rating Curve= 0 ,0
Exp/Cntr=0.3,0.1

Type RM Length L Ch R = 1 ,6308.2  ,204,203.6,203.3
XS GIS Cut Line= 4
     1650420.061      210025.167     1650429.382      210399.547
     1650426.275      210623.243     1650528.802      210958.787
#Sta/Elev= 30
    10.1  1105.8    20.2 1099.92    30.4  1099.7    70.9  1074.9   121.5 1046.83
   131.6 1046.67   222.7  978.17   232.8  978.21   313.8  923.19   323.9  917.62
     334  917.53   364.4  912.19   374.5  907.51   423.1  874.24   442.3  867.09
   452.3  865.42   462.3  865.95   500.9  871.17   618.3  876.22   628.3     879
   638.3  884.25   648.3  885.53   658.4  890.31   738.6  941.21   758.6  951.48
   768.6  953.34   858.9  1009.7   878.9  1015.9     919 1039.78   949.1 1049.52
#Mann= 3 , 0 , 0
       0      .1       0   442.3    .045       0   462.3      .1       0
Bank Sta=442.3,462.3
XS Rating Curve= 0 ,0
Exp/Cntr=0.3,0.1

Type RM Length L Ch R = 1 ,6104.5  ,213.7,223,232.3
XS GIS Cut Line= 3
     1650165.513      210085.113     1650225.344      210395.023
     1649900.356       211019.54
#Sta/Elev= 30
     9.9 1110.47    29.6 1095.29    39.5 1093.55    49.3 1086.87    88.8 1050.48
   138.1  995.32     148  986.71   157.8  982.35   207.1  938.27   246.6  917.32
   256.5  916.61   276.2  907.91   305.8  904.09   345.3  878.71  380.13  863.17
   384.8  862.24  400.28  863.39   503.4   869.6   562.7  884.73   652.4  901.07
   662.4  903.71   682.3  913.59   702.2  919.13   801.8  978.66   821.7  984.48
   841.7  995.86   931.3 1053.87   941.3 1059.43   951.2 1061.02  1060.8 1128.33
#Mann= 3 , 0 , 0
     9.9      .1       0  380.13    .045       0  400.28     .08       0
Bank Sta=380.13,400.28
XS Rating Curve= 0 ,0
Exp/Cntr=0.3,0.1

Type RM Length L Ch R = 1 ,5881.6  ,180.2,179.7,179.3
XS GIS Cut Line= 4
     1650087.624       210112.16     1650033.254      210376.245
     1649968.009      210544.017     1649703.923       210910.63
#Sta/Elev= 30
      10 1063.93    89.9  999.17    99.9  992.94   109.8  990.38   199.7  915.83
   209.7  914.94   229.7  903.57   239.7  900.85   259.6  900.22   269.6   897.2
   299.6  876.48   319.6   868.3   329.6  860.15  334.51  858.63   339.6  857.18
  354.73  857.81   379.6  860.83   449.6  862.95   519.9   883.7     540  885.55
   580.2   901.5   620.3  921.93   640.4  935.02   660.5  941.53   700.7  968.44
   750.9 1006.64     781 1021.72   851.3 1069.12   881.4 1092.88   901.5 1101.73
#Mann= 3 , 0 , 0
      10      .1       0  334.51    .045       0  354.73      .1       0
Bank Sta=334.51,354.73
XS Rating Curve= 0 ,0
Exp/Cntr=0.3,0.1

Type RM Length L Ch R = 1 ,5701.8  ,446.2,441.9,437.5
XS GIS Cut Line= 4
      1649942.29      210091.002     1649880.887      210267.723
      1649783.54      210531.308      1649573.87      210883.254
#Sta/Elev= 30
     9.8 1021.26    19.7 1017.61   108.3  954.11     128  947.41   197.1  902.44
   207.2  897.43   237.3  894.91   247.3  891.64   297.5   855.6   302.1  854.23
   307.5  852.67  322.27     853   377.8  857.43     438  858.63     448  860.17
     458  864.71   488.1  882.39     538   916.2     548  917.99     578  936.72
     598  951.33   637.9  988.29   647.9  994.58   657.9  996.59   737.9 1050.49
   757.8  1067.2   777.8 1076.03   807.8 1100.98   867.7 1144.82   877.7 1148.54
#Mann= 3 , 0 , 0
     9.8      .1       0   302.1    .045       0  322.27      .1       0
Bank Sta=302.1,322.27
XS Rating Curve= 0 ,0
Exp/Cntr=0.3,0.1

Type RM Length L Ch R = 1 ,5260    ,333.3,312.2,291
XS GIS Cut Line= 4
     1649534.931      210026.603     1649428.599      210216.804
     1649388.163      210442.948     1649398.646      210847.311
#Sta/Elev= 30
     9.9  954.82    19.8  947.63    29.7  945.54    39.6  940.36    69.3  921.04
     109  891.64   138.7  874.24   148.6   873.7   178.3  863.32     208  858.33
   267.8  856.19   297.8  859.67   347.8  847.41   357.7  846.51   367.7  846.18
   377.7  847.12   397.7   851.1   447.6  881.99   467.9  889.29   548.8  945.07
   558.9  950.84     569  952.53   649.9 1017.16     660 1023.59   670.1 1025.19
   700.4 1047.83   720.7 1060.82   761.1  1083.5   771.2 1084.57   852.1 1132.87
#Mann= 3 , 0 , 0
       0     .08       0   357.7    .045       0   377.7     .08       0
Bank Sta=357.7,377.7
XS Rating Curve= 0 ,0
Exp/Cntr=0.3,0.1

Type RM Length L Ch R = 1 ,4947.8  ,255.9,258.1,260.3
XS GIS Cut Line= 4
     1648948.372       210055.02     1649065.345      210256.799
     1649201.326      210430.796      1649359.24      210835.816
#Sta/Elev= 30
     9.7  967.76    19.4  955.88    29.2   949.1    38.9  944.94    48.6   938.6
    58.3   935.7   116.6  908.78   165.2  888.67   174.9  886.88   233.2  864.47
   283.4  848.94   363.8  838.96   373.8  838.52   383.8  838.91   403.9  842.32
     434  853.05   464.2  861.55   514.7  883.03   524.8  887.99   555.2  905.78
   575.4  912.42     636  951.97   676.5  980.08   696.7  987.62   787.7 1051.53
   797.8 1054.44   807.9 1059.58   828.1 1073.53   858.4  1097.7   888.8  1113.8
#Mann= 3 , 0 , 0
       0      .1       0   363.8    .045       0   383.8     .08       0
Bank Sta=363.8,383.8
XS Rating Curve= 0 ,0
Exp/Cntr=0.3,0.1

Type RM Length L Ch R = 1 ,4689.7  ,364.8,358.2,351.6
XS GIS Cut Line= 4
     1648676.523      210147.126     1648860.234      210388.746
     1649000.014      210606.403     1649274.471      210922.905
#Sta/Elev= 30
    10.1 1066.26    20.2 1059.97    40.5 1052.99    91.1 1021.27   121.4 1002.13
   141.6  983.75   151.8  977.37   212.5  965.41   222.6  956.96   242.8  908.56
   273.2  884.03   303.5  865.16   323.4  858.67   353.3  841.24   363.2  838.88
   412.9  837.53   422.9  837.01   432.9  837.07   462.7  838.15   532.4  858.96
   582.2  870.36   691.9   928.8   721.8  947.74   731.8   950.5   741.7   959.1
   841.5 1019.26   861.4 1035.89   911.3 1057.21   961.2 1071.56   981.1 1081.09
#Mann= 3 , 0 , 0
       0      .1       0   412.9    .045       0   432.9     .08       0
Bank Sta=412.9,432.9
XS Rating Curve= 0 ,0
Exp/Cntr=0.3,0.1

Type RM Length L Ch R = 1 ,4331.6  ,294.9,295,295.1
XS GIS Cut Line= 4
     1648414.196      210453.681      1648532.01      210565.505
     1648751.665       210765.19     1649099.117      210976.857
#Sta/Elev= 30
     9.6  915.77    28.7  912.54    66.9  901.45   152.9  868.63   162.4  866.47
   172.3  866.58     202  854.88   231.7  846.71   261.4  832.19   271.2  829.43
   281.2  828.84   291.2  828.98     390  831.47   409.8  835.51   429.6  842.48
   469.2  853.29     499  859.07   518.8  866.73   528.8  874.17   538.7  879.18
   578.4  904.29   608.1  919.87     628  933.74   647.8  943.82   667.7  951.74
   747.1  975.47   766.9  975.35   776.8  979.97   816.5  983.34   866.1  991.41
#Mann= 3 , 0 , 0
       0      .1       0   271.2    .045       0   291.2      .1       0
Bank Sta=271.2,291.2
XS Rating Curve= 0 ,0
Exp/Cntr=0.3,0.1

Type RM Length L Ch R = 1 ,4036.5  ,369.2,370,370.8
XS GIS Cut Line= 4
     1648200.532      210547.533     1648382.246      210821.102
     1648575.941      210998.822     1648813.567      211312.329
#Sta/Elev= 30
      10  1029.7    69.7  998.24   119.4  968.88   228.9  907.82   238.9  902.97
   248.8  900.48   258.8  894.65   288.6  872.37   308.5  861.18   358.8  838.18
   409.4  823.72   419.4  823.32   429.4  823.41   490.2  824.91   500.3  827.51
   530.6  840.42   550.9  846.67   591.3  851.52   621.6  866.55   651.8  885.97
   702.2  912.83   722.4  919.67   742.6  930.64   782.9  952.91   803.1  967.08
   843.5  987.73   863.6   994.7   914.1 1020.49   934.2 1035.05   984.7 1061.41
#Mann= 3 , 0 , 0
       0      .1       0   409.4    .045       0   429.4      .1       0
Bank Sta=409.4,429.4
XS Rating Curve= 0 ,0
Exp/Cntr=0.3,0.1

Type RM Length L Ch R = 1 ,3666.6  ,257.6,254.4,251.2
XS GIS Cut Line= 4
     1647946.783      210731.207      1648074.73      211032.769
     1648328.331      211280.379     1648674.527      211533.499
#Sta/Elev= 30
     9.9 1097.85    39.7 1079.64    69.5 1057.69    99.3 1044.22   198.5  985.17
   218.4  978.05   297.8  935.05   317.7  919.91   337.7  911.62     439  841.57
   469.4  818.28   479.6  814.59   489.6  814.55   499.6  814.75   550.4  816.35
   560.5  818.67   590.9  831.57   631.4  837.82   661.8  849.72   761.8  899.96
   781.8  913.26   831.6  939.11   851.6  945.32   881.5  959.19   951.3 1000.57
   991.2 1027.07  1041.1 1055.57    1071 1066.62    1081 1068.09  1110.9  1082.9
#Mann= 3 , 0 , 0
       0      .1       0   479.6    .045       0   499.6      .1       0
Bank Sta=479.6,499.6
XS Rating Curve= 0 ,0
Exp/Cntr=0.3,0.1

Type RM Length L Ch R = 1 ,3412.1  ,224.4,236.8,249.3
XS GIS Cut Line= 4
     1647674.607      211051.541     1647944.906      211279.897
     1648110.348      211404.561     1648440.067      211627.092
#Sta/Elev= 30
    10.1 1100.47    20.2 1091.86    30.3 1079.76   101.1 1031.26   121.3 1014.37
   141.5  993.49   151.6  986.35   212.3  951.21   252.7  933.14   262.9  930.04
   283.1  918.73   343.7     881   363.7  863.96   442.5   810.2   452.5  809.47
   462.5  809.87   511.7  812.64   570.9  827.83   590.8  834.82   640.6  857.63
   660.4  870.68   690.3  886.42     740  917.16   749.9   924.5   759.9  934.81
   839.5   989.3   859.3 1007.67   889.2 1022.14   938.9 1051.68   958.8 1065.54
#Mann= 3 , 0 , 0
       0      .1       0   442.5    .045       0   462.5      .1       0
Bank Sta=442.5,462.5
XS Rating Curve= 0 ,0
Exp/Cntr=0.3,0.1

Type RM Length L Ch R = 1 ,3175.3  ,187.2,185.3,183.4
XS GIS Cut Line= 4
     1647633.181      211073.742       1647799.4      211389.091
     1647895.714       211600.36     1648225.044      211861.339
#Sta/Elev= 30
     9.9 1115.22    19.8 1111.84    29.7  1104.9    79.2  1059.5   128.7 1018.21
   158.4  1002.6   188.1  979.08   247.6  942.52   257.5  936.75   267.4  935.23
   277.3  930.63   297.1  918.68   376.7  858.73   396.9  850.26   427.1  828.13
   447.3  810.67   457.5  806.74   467.5  806.42   477.5  806.96   538.2  810.27
   598.7  819.77   648.7   835.4   698.7  861.74   718.7  875.52   798.8   920.5
   818.8  936.09   838.8  944.38   898.8  975.49   918.8  988.63  1008.9 1027.26
#Mann= 3 , 0 , 0
       0      .1       0   457.5    .045       0   477.5      .1       0
Bank Sta=457.5,477.5
XS Rating Curve= 0 ,0
Exp/Cntr=0.3,0.1

Type RM Length L Ch R = 1 ,2990    ,187.8,188.5,189.2
XS GIS Cut Line= 4
     1647598.887      211057.804     1647595.337       211416.35
     1647781.192      211755.631     1647783.485      212186.693
#Sta/Elev= 30
      10 1123.49    29.9 1123.67    39.8 1121.18    59.8 1109.95   119.5 1063.46
   129.5 1061.14   139.4  1055.8   219.1   998.7     239   991.2   318.7  922.92
   338.6  915.94   358.6  903.16   447.8  835.35   457.8   835.1   507.3  799.84
   517.3  797.89   527.3  799.47     676   814.8   715.7  824.52   745.4  836.54
   805.6  866.05   825.6  871.54   905.8  917.89   925.9  923.66     986  959.21
  1006.1   973.1  1026.1  979.57  1106.3 1030.55  1136.4    1043  1176.5 1068.73
#Mann= 3 , 0 , 0
       0      .1       0   507.3    .045       0   527.3      .1       0
Bank Sta=507.3,527.3
XS Rating Curve= 0 ,0
Exp/Cntr=0.3,0.1

Type RM Length L Ch R = 1 ,2801.5  ,126.7,128.5,130.3
XS GIS Cut Line= 4
     1647553.438      211100.474     1647470.717      211574.663
     1647572.079      211771.563     1647696.743      212133.903
#Sta/Elev= 30
      10 1089.35    30.1 1072.32    50.1 1060.18    90.3 1045.86   140.4 1019.85
   170.5  996.11   190.5  986.87   220.6  964.06   250.7  945.28   270.8  934.42
   290.8  929.09   320.9  912.46   330.9  904.75     351  882.34     371  866.04
   381.1   860.1   391.1  858.97   451.3  816.86   481.4  807.04   551.9  793.05
   561.9  792.34   571.9  792.79   682.7  799.27   743.1  811.82   833.9  867.33
   854.1  874.56   954.9  943.37   975.1  951.16  1055.7 1001.48    1086 1014.66
#Mann= 3 , 0 , 0
       0      .1       0   551.9    .045       0   571.9      .1       0
Bank Sta=551.9,571.9
XS Rating Curve= 0 ,0
Exp/Cntr=0.3,0.1

Type RM Length L Ch R = 1 ,2672.9  ,339.6,338.4,337.3
XS GIS Cut Line= 4
     1647518.375      211079.997      1647375.18      211658.549
      1647446.25      211825.156     1647640.819      212140.894
#Sta/Elev= 30
    10.1 1071.78    80.8 1040.81   111.1 1032.07   141.4 1017.37   191.9  975.38
   212.1  967.04   242.4  947.34   282.9  926.17   303.1   917.1   313.2  916.05
   333.4   906.1     394  867.27   414.2  859.78   454.6  835.48   484.9   826.3
   525.3  822.17   575.8  806.99   616.1  803.05  650.53   791.6   656.4  790.17
  671.72  791.43   706.7  797.51   767.1  795.76   827.3  807.59   847.3  818.42
   867.4  824.55   997.7  893.69  1107.9  962.26    1128  970.33    1148  982.27
#Mann= 3 , 0 , 0
    10.1      .1       0  650.53    .045       0  671.72      .1       0
Bank Sta=650.53,671.72
XS Rating Curve= 0 ,0
Exp/Cntr=0.3,0.1

Type RM Length L Ch R = 1 ,2334.5  ,414.6,414.4,414.3
XS GIS Cut Line= 4
     1646846.294       211458.95     1647048.642      211760.697
     1647185.001      212042.102     1647311.339      212399.691
#Sta/Elev= 30
    10.1  1032.1    60.6   982.8    70.6  975.63    80.7  972.79     111  938.59
   151.4  900.42   201.8  861.43   211.9  860.68   282.6  823.19     333  802.12
   383.5  792.73   433.9  791.89   454.2  784.01   464.2  782.57   474.2  782.65
   585.2  789.32   615.5  796.19   655.8  825.22     696  858.15     706  859.55
   715.9  865.77   815.7  944.05   825.7  944.89   885.6  992.38   915.5  1018.4
   925.5  1025.5   935.5 1027.98   995.4    1078  1035.3  1101.2  1055.3 1107.64
#Mann= 3 , 0 , 0
       0      .1       0   454.2    .045       0   474.2     .08       0
Bank Sta=454.2,474.2
XS Rating Curve= 0 ,0
Exp/Cntr=0.3,0.1

Type RM Length L Ch R = 1 ,1920.1  ,218.4,214,209.5
XS GIS Cut Line= 4
     1646473.251      211649.798     1646682.921      211949.326
      1646772.78      212133.037     1647050.343      212466.512
#Sta/Elev= 30
     9.9  972.04    29.6   958.6    49.4  949.47    88.9  920.64   118.6   901.2
   138.3     883     168  866.64   207.5  849.23   296.4  823.09   326.1  817.24
   404.6  790.67   443.5  786.89   462.7  779.03   472.7  778.07   482.7  780.61
   521.4  785.71   550.7   793.8   600.4  795.57   610.5  799.72   630.7  813.46
   660.9   825.5   721.5  838.38     782  859.89   842.6  885.39   862.7  887.76
   872.8  891.59   903.1   904.4   983.8  949.05   993.9  953.38    1004  955.03
#Mann= 3 , 0 , 0
       0      .1       0   462.7    .045       0   482.7     .06       0
Bank Sta=462.7,482.7
XS Rating Curve= 0 ,0
Exp/Cntr=0.3,0.1
